--- CARNEYFK.prj (project) ---

Proj Title=CARNEYFK
Current Plan=p01
Default Exp/Contr=0,0
English Units
Geom File=g01
Flow File=f01
Plan File=p01
BEGIN DESCRIPTION:
---------- MODELED AS PART OF WVEMD CTP PROGRAM, 2023----------
Stream Name: Carney Fork
Flood Zone:  AFH
Wetzel County, WV
HEC-RAS Version: RAS 6.3
Vertical Datum: NAVD88
Projection: NAD 1983 StatePlane West Virginia S FIPS 4702 (US Feet)
Terrain: 1-meter West Virginia FEMA R3 South Central (collected 2018-2020)
Land Use: 2019 NLCD
Hydrologic Method:
WV SIR2010-5033 regression equations
Additional Model Notes:
None
END DESCRIPTION:
DSS Export Rating Curves= 0
DSS Export Rating Curve Sorted= 0
DSS Export Volume Flow Curves= 0
DXF OffsetX= 0
DXF OffsetY= 0
DXF ScaleX= 0
DXF ScaleY= 0

--- CARNEYFK.p01 (plan) ---

Plan Title=Floodplain
Program Version=6.30
Short Identifier=Floodplain
Geom File=g01
Flow File=f01
Subcritical Flow
K Sum by GR= 0
Std Step Tol= 0.01
Critical Tol= 0.01
Num of Std Step Trials= 20
Max Error Tol= 0.3
Flow Tol Ratio= 0.001
Split Flow NTrial= 30
Split Flow Tol= 0.02
Split Flow Ratio= 0.02
Log Output Level= 0
Friction Slope Method= 1
Unsteady Friction Slope Method= 2
Unsteady Bridges Friction Slope Method= 1
Parabolic Critical Depth
Global Vel Dist= 0 , 0 , 0
Global Log Level= 0
CheckData=True
Encroach Param=-1 ,0,0, 0
Mapping Interval=1HOUR
Computation Time Step Use Courant=        0
Computation Time Step Use Time Series=    0
Computation Time Step Count To Double=0
Computation Time Step Max Doubling=0
Computation Time Step Max Halving=0
Computation Time Step Residence Courant=0
Run HTab= 0
Run UNet= 0
Run Sediment= 0
Run PostProcess= 0
Run WQNet= 0
Run RASMapper= 0
UNET Theta= 0
UNET Theta Warmup= 0
UNET ZTol= 0
UNET ZSATol= 0
UNET MxIter= 0
UNET Max Iter WO Improvement= 0
UNET MaxInSteps= 0
UNET DtIC= 0
UNET DtMin= 0
UNET MaxCRTS= 0
UNET WFStab= 0
UNET SFStab= 0
UNET WFX= 1
UNET SFX= 1
UNET Gravity=32.17405
UNET 1D Methodology=Finite Difference
UNET DSS MLevel= 1
UNET Pardiso=0
UNET DZMax Abort= 0
UNET Use Existing IB Tables= 0
UNET Froude Reduction=False
UNET Froude Limit= 0
UNET Froude Power= 0
UNET D1 Cores= 0
UNET WindReference=Eulerian
UNET WindDragFormulation=Hsu (1988)
UNET D2 Coriolis=0
UNET D2 Cores= 0
UNET D2 Theta= 1
UNET D2 Theta Warmup= 1
UNET D2 Z Tol= 0.01
UNET D2 Volume Tol= 0.01
UNET D2 Max Iterations= 20
UNET D2 Equation= 0
UNET D2 RampUpFraction=0.1
UNET D2 TimeSlices= 1
UNET D2 Turbulence Formulation=Non-Conservative (original)
UNET D2 Eddy Viscosity=0.3
UNET D2 Transverse Eddy Viscosity=0.1
UNET D2 Smagorinsky Mixing=0
UNET D2 BCVolumeCheck=0
UNET D2 Cores=0
UNET D2 SolverType=PARDISO (Direct)
UNET D2 Minimum Iterations= 3
UNET D2 Maximum Iterations= 30
UNET D2 Restart Number= 10
UNET D2 Relaxation Coeff=1.3
UNET D2 SOR Precondition Iterations= 10
UNET D2 ILUT Maximum Fill= 8
UNET D2 ILUT Tolerance=1E-08
UNET D2 Convergence Tolerance=0.00001
UNET D1D2 MaxIter= 0
UNET D1D2 ZTol=0.01
UNET D1D2 QTol=0.1
UNET D1D2 MinQTol=1
Write IC File= 0
Write IC File at Fixed DateTime=0
Write IC File at Sim End=0
Echo Input=False
Echo Parameters=False
Echo Output=False
Write Detailed= 0
HDF Write Warmup=0
HDF Write Time Slices=0
HDF Flush=0
HDF Compression= 1
HDF Chunk Size= 1
HDF Spatial Parts= 1
HDF Use Max Rows=0
HDF Fixed Rows= 1
Calibration Method= 0
Calibration Iterations= 20
Calibration Max Change=0.05
Calibration Tolerance=0.2
Calibration Maximum=1.5
Calibration Minimum=0.5
Calibration Optimization Method= 1
WQ AD Non Conservative
WQ ULTIMATE=-1
WQ Max Comp Step=1HOUR
WQ Output Interval=15MIN
WQ Output Selected Increments= 0
WQ Output face flow=0
WQ Output face velocity=0
WQ Output face area=0
WQ Output face dispersion=0
WQ Output cell volume=0
WQ Output cell surface area=0
WQ Output cell continuity=0
WQ Output cumulative cell continuity=0
WQ Output face conc=0
WQ Output face dconc_dx=0
WQ Output face courant=0
WQ Output face peclet=0
WQ Output face adv mass=0
WQ Output face disp mass=0
WQ Output cell mass=0
WQ Output cell source sink temp=0
WQ Output nsm pathways=0
WQ Output nsm derived pathways=0
WQ Create Restart=0
WQ Fixed Restart=0
WQ System Summary=0
WQ Write To DSS=0
Sorting and Armoring Iterations= 10
XS Update Threshold= 0.02
Bed Roughness Predictor= 0
Hydraulics Update Threshold= 0.02
Energy Slope Method= 1
Volume Change Method= 1
Sediment Retention Method= 0
Sediment TS Multiplier= 1
Warm Up Method= 0
XS Weighting Method= 0
Number of US Weighted Cross Sections= 1
Number of DS Weighted Cross Sections= 1
Upstream XS Weight=0
Main XS Weight=1
Downstream XS Weight=0
Number of DS XS's Weighted with US Boundary= 1
Upstream Boundary Weight= 1
Weight of XSs Associated with US Boundary= 0
Number of US XS's Weighted with DS Boundary= 1
Downstream Boundary Weight= 0.5
Weight of XSs Associated with DS Boundary= 0.5
Percentile Method= 0
Sediment Output Level= 3
Mass or Volume Output= 0
Output Increment Type= 1
Profile and TS Output Increment= 1
Transport Output Increment 1
XS Output Flag= 0
XS Output Increment= 10
Read HDF5 Sediment Hotstart= 0
Sediment Hotstart Type= 0
Write Gradation File= 0
Read Gradation Hotstart= 0
Write HDF5 File= 1
Write Binary Output= 1
Write DSS Sediment File= 0
DSS Sediment Output Type= 1
SV Curve= 0
Specific Gage Flag= 0
Subcell Erosion Methods= 0
Subcell Deposition Methods= 0
Advection Scheme= 1
Matrix Solver= 0
Implicit Weighting Factor= 1
Maximum Outer Loop Convergence Iterations= 5
Convergence Maximum Absolute= 0.001
Convergence RMSE= 0.0001
Grain Fractions Max Abs Error= 0.001
Max Subgrid Regions= 1
Max Subgrid Length Scale= 3.402823E+38
Initial Layer Thickness= 3.402823E+38
Min Layer Thickness= 3.402823E+38
Max Layer Thickness= 3.402823E+38
Number of Layers= 5

--- CARNEYFK.f01 (steady flow) ---

Flow Title=Flow
Program Version=4.00
Number of Profiles=1
Profile Names=F01pct
River Rch & RM=CARNEYFK,Main,19960
     668
River Rch & RM=CARNEYFK,Main,18490
     753
River Rch & RM=CARNEYFK,Main,17492
     838
River Rch & RM=CARNEYFK,Main,14555
     986
River Rch & RM=CARNEYFK,Main,13446
    1120
River Rch & RM=CARNEYFK,Main,9493
    1500
River Rch & RM=CARNEYFK,Main,3000
    1700
Boundary for River Rch & Prof#=CARNEYFK,Main      ,1
Up Type=0
Dn Type=3
Dn Slope=0.013989

--- CARNEYFK.g01 (geometry) ---

Geom Title=Geometry
Program Version=6.31

River Reach=CARNEYFK        ,Main
Reach XY= 30
     1653558.946      429044.449     1654913.408      429998.897
     1655633.702      430279.815     1656040.444      430737.694
     1656986.481      430860.154     1657204.487      431326.108
     1657508.955      431575.065     1657870.952      431657.154
     1658316.047      432152.376     1658973.429       432524.13
       1659285.5      433262.631      1659330.07      433733.093
     1659560.457      434026.782     1659535.265      434664.543
     1659900.869      434973.735     1660049.866      435315.869
     1660673.847      435765.015     1660706.144      435972.578
     1661187.802      436528.089     1661515.511      436737.589
      1661412.16      437389.131     1661756.122      437954.527
      1661607.47      438670.713     1661900.512      438992.332
     1662560.295      439179.338     1662600.153      440149.711
     1662709.198      440370.056     1663408.337      440860.131
     1663502.592      441562.279     1664308.157      441644.187

Type RM Length L Ch R = 1 ,19960   ,96.5,96.4,96.1
XS GIS Cut Line= 4
1653297.32146105429063.8311864671653508.44334849429085.957497814
1653724.17488412428981.7794485551653779.49066249428782.642646433
#Sta/Elev= 30
       0 1177.78      43 1159.46    51.1 1155.07    63.1 1145.67    71.2 1140.18
    83.2 1135.06    87.3 1134.18   111.4 1133.36   119.4  1132.3   151.6 1123.34
   175.8 1118.29   212.3    1116   238.6 1115.17   265.2 1111.66  271.25 1110.31
     276 1109.65   279.9 1110.32     291 1114.57   314.1 1120.26   335.1  1121.4
   389.6 1122.76   429.6 1126.23   461.4 1131.62   482.2 1132.83     495 1139.79
   511.3 1147.45   550.3 1157.54   594.3 1173.22   631.6 1182.19   658.5  1186.7
#Mann= 8 ,-1,0
       0      .1       0      90     .05       0  271.25    .045       0
   279.9     .05       0  302.28     .06       0  402.28     .07       0
  491.85     .06       0  591.85      .1       0
Bank Sta=271.25,279.9
XS Rating Curve= 0 ,0
Exp/Cntr(USF)=0,0
Exp/Cntr=0.3,0.1

Type RM Length L Ch R = 1 ,19863   ,449.7,452.7,451.2
XS GIS Cut Line= 6
1653515.45643763429363.5793538061653521.14186466429186.383544683
1653645.27368816429120.0535626581653679.38625034429059.409007664
 1653751.4016594428975.0751733761653773.19579635428880.318056198
#Sta/Elev= 30
       0 1169.31    31.1 1159.66    51.1 1154.29    72.8 1147.23    75.1 1146.23
    83.1 1141.21   103.1 1126.57   111.1 1121.43   119.1 1117.92   126.5 1115.91
   143.1  1114.5   177.3 1113.09   225.2  1112.5   246.6 1111.64  283.85 1108.22
   285.9 1108.07  290.96 1108.22   356.6 1113.95   410.1 1121.15   454.6 1125.95
   483.9 1130.72   492.4  1131.2   505.3 1130.07   513.5 1131.76   521.7 1136.23
   529.9 1139.57   541.4 1141.87   558.7  1147.9   578.1 1152.91   595.8  1158.5
#Mann= 8 ,-1,0
       0      .1       0     120     .05       0  283.85    .045       0
  290.96     .05       0  378.14      .1       0  407.72     .07       0
  528.61     .06       0  595.85      .1       0
Bank Sta=283.85,290.96
XS Rating Curve= 0 ,0
Exp/Cntr(USF)=0,0
Exp/Cntr=0.3,0.1

Type RM Length L Ch R = 1 ,19411   ,593.9,594.9,591.6
XS GIS Cut Line= 3
1653775.11718358429551.8249431181653923.38919958429328.774514422
1654139.39971151429025.417654854
#Sta/Elev= 30
       0 1183.95    49.3 1167.77    60.8  1164.9    92.5 1151.63   115.6 1143.66
   153.1 1131.71   210.8 1115.98   242.6 1110.26     273  1106.8   302.5 1104.58
   327.1 1104.36   334.5 1103.29   340.81104.363   354.6 1110.54   374.6 1126.19
   406.2 1138.83   420.4 1145.25   429.1 1150.71     432 1151.47   452.1 1152.69
     455 1153.83   463.6 1160.57   466.4 1162.04     476 1164.96   528.4 1184.05
   552.9    1195   567.7 1198.94   579.4 1204.48     607 1215.28   640.2 1229.87
#Mann= 4 ,-1,0
       0     .05       0   327.1    .045       0   340.8     .05       0
  347.84      .1       0
Bank Sta=327.1,340.8
XS Rating Curve= 0 ,0
Exp/Cntr(USF)=0,0
Exp/Cntr=0.3,0.1

Type RM Length L Ch R = 1 ,18816   ,325.2,325.9,324.2
BEGIN DESCRIPTION:
Structure XS 4
END DESCRIPTION:
XS GIS Cut Line= 6
1654234.47028435 429978.743852161654355.21249695429752.852899737
1654392.71865552429657.8711343181654425.54142452429584.000547147
1654470.09415695429502.7021533171654502.65208381429449.356407223
#Sta/Elev= 30
       0 1213.81    52.4 1195.04    64.9 1189.14    97.4 1177.52   115.2 1173.54
   129.9 1166.25   174.9 1148.59   189.1 1140.56   197.5 1138.87   215.7 1137.93
   269.4 1125.32   290.9 1109.95   303.3 1103.87   316.7 1101.78   342.5 1099.91
   386.1 1098.15   394.7  1097.3  399.371098.188   422.4 1112.94   434.1 1119.18
   461.3 1127.48   481.7 1134.89   488.7 1138.45   497.8 1145.29     516 1146.71
   519.4 1148.69   529.7 1158.75   534.3 1161.89   548.4 1165.93   594.3  1185.5
#Mann= 5 ,-1,0
       0     .05       0  276.14     .06       0   386.1    .045       0
  399.37     .06       0  519.09      .1       0
Bank Sta=386.1,399.37
XS Rating Curve= 0 ,0
Exp/Cntr(USF)=0,0
Exp/Cntr=0.3,0.1

Type RM Length L Ch R = 1 ,18490   ,37,37.5,38.2
BEGIN DESCRIPTION:
Structure XS 3
END DESCRIPTION:
XS GIS Cut Line= 6
  1654256.933606429991.6521257531654548.01837847429969.300836288
1654607.76970894 429918.33631531 1654666.7556892429788.665067662
1654640.51111815 429715.283156081654643.30741537429505.497807514
#Sta/Elev= 30
       0 1208.47    35.7 1195.71    55.3 1187.92    69.6 1183.73    99.5 1170.49
   123.5 1158.69   135.6 1156.15   139.6 1154.42   183.7 1133.08   187.7 1131.76
   199.8 1130.67   215.8 1124.23   251.9 1114.59     288 1101.98   305.4 1100.68
   381.6 1100.03     406 1097.27   492.8 1095.27     497 1094.29   502.91095.279
   554.7 1096.79   568.5 1097.82   607.8 1108.69   635.8 1114.87   679.8 1133.06
   695.8 1133.65   699.8 1134.43   709.8 1144.22   715.8 1148.02   802.8 1185.96
#Mann= 6 ,-1,0
       0     .05       0     110      .1       0     210     .05       0
  479.63      .1       0   492.8    .045       0   502.9      .1       0
Bank Sta=492.8,502.9
XS Rating Curve= 0 ,0
Exp/Cntr(USF)=0,0
Exp/Cntr=0.3,0.1

Type RM Length L Ch R = 1 ,18452   ,430.2,434.9,429.9
BEGIN DESCRIPTION:
Structure XS 2
END DESCRIPTION:
XS GIS Cut Line= 6
1654266.70606017430026.5591570351654555.68068431430004.871406402
 1654635.9807559429943.1021205581654702.35968994429805.365832424
1654671.68233258429705.8428470811654672.19054904429516.821878619
#Sta/Elev= 30
       0 1207.61    21.5 1199.41    38.4 1194.47    53.6 1185.25    89.7 1170.02
   101.7 1161.91   113.7 1159.87   145.8 1142.28   161.9 1130.93   165.9 1129.56
   177.9 1128.91     214 1112.12     226 1107.74   242.1 1103.77   324.5 1099.96
   512.5 1095.87524.74271094.832   530.9 1093.65536.54271094.825   622.9 1100.75
   646.3  1103.9     651 1105.39   674.9 1117.33   710.8  1130.6   714.6 1131.43
   734.6  1131.6   738.6 1133.61   750.7 1143.02   806.6 1170.94   838.3 1184.74
#Mann= 8 ,-1,0
       0     .05       0     100      .1       0     200     .05       0
  520.36      .1       0524.7427    .045       0536.5427      .1       0
  622.54     .06       0  719.26      .1       0
Bank Sta=524.7427,536.5427
XS Rating Curve= 0 ,0
Exp/Cntr(USF)=0,0
Exp/Cntr=0.3,0.1

Type RM Length L Ch R = 1 ,18017   ,512,525.5,523.5
BEGIN DESCRIPTION:
Structure XS 1
END DESCRIPTION:
XS GIS Cut Line= 6
1654842.14490801430294.3824913351654939.00560668430126.073772833
1654988.99041484430054.7553459261655039.54264943429944.412344548
1655063.47265387429898.4836110251655215.51784892429764.026268587
#Sta/Elev= 30
       0 1199.47    78.2 1172.21    93.6 1168.64   102.8 1165.47   154.1 1139.43
   181.6 1130.72   205.9 1119.52   230.3 1107.29   254.7 1093.07   276.5 1088.72
   318.9 1089.73   330.6 1089.24   336.5  1087.3   339.6 1087.17   348.7  1089.2
   378.9 1098.03   420.6 1112.16   425.1 1114.19   435.6 1121.38   441.6 1122.43
   456.3 1122.76   463.4 1128.07   469.5 1131.36   481.6 1136.27   515.8 1153.08
   541.9  1163.8   560.1 1168.97   583.5 1177.39     632 1197.85   657.4 1202.73
#Mann= 6 ,-1,0
       0     .05       0      80      .1       0   330.6    .045       0
   348.7      .1       0  422.68     .06       0  554.47      .1       0
Bank Sta=330.6,348.7
XS Rating Curve= 0 ,0
Exp/Cntr(USF)=0,0
Exp/Cntr=0.3,0.1

Type RM Length L Ch R = 1 ,17492   ,488,497.9,491.9
XS GIS Cut Line= 6
1655218.79704183430456.3047396691655276.57087642430378.882978499
1655333.21315159430309.1524749251655502.45297059430124.348710671
1655552.06507608 430050.885931091655593.93277451429964.184004754
#Sta/Elev= 30
       0  1169.9    17.9  1164.3    77.9 1140.28   102.2 1132.83   126.4 1127.72
   160.5 1108.63   190.7 1097.83   196.6 1096.24   299.3 1082.69   307.8 1081.32
     3171082.696   350.3  1085.4   360.9 1087.61   377.2 1094.97   393.4 1099.53
   409.8 1106.19   421.7 1108.27   432.4  1114.4   456.1 1124.79   465.8 1126.56
   485.1 1126.72   487.1 1127.41   489.9  1128.5   499.5 1134.91   525.7  1141.8
   554.9 1157.88   568.3 1163.22     586  1167.5   608.2 1174.87     622 1175.95
#Mann= 7 ,-1,0
       0      .1       0      40     .05       0      50      .1       0
   299.3    .045       0     317      .1       0  432.03     .06       0
  555.67      .1       0
Bank Sta=299.3,317
XS Rating Curve= 0 ,0
Exp/Cntr(USF)=0,0
Exp/Cntr=0.3,0.1

Type RM Length L Ch R = 1 ,16994   ,403.6,416.6,411
XS GIS Cut Line= 6
  1655577.108005430668.0129776751655650.18266201430597.216531336
1655711.43549226430524.3154304181655795.30277859430365.680249006
1655861.43584843430214.7317320111655912.38784626430132.751252919
#Sta/Elev= 30
       0 1165.38   102.6 1126.45     115 1123.48   135.8 1113.95   163.2 1103.89
   210.6 1093.07   238.3 1084.12   261.7  1080.8     311 1077.55   321.2 1076.13
   332.9 1077.56   354.1 1078.17   360.2 1079.91     372 1087.67   381.1 1095.56
   399.4 1113.59   408.1  1123.1   411.6 1125.56   416.8 1126.93     430 1127.38
   434.1 1128.41   442.8 1134.52   454.4 1139.79   482.2 1157.89   526.2 1178.35
     542 1187.21   576.7 1209.47     591 1215.96   622.2 1232.94   637.9 1240.03
#Mann= 5 ,-1,0
       0      .1       0     311    .045       0   332.9      .1       0
  426.51     .06       0  492.56      .1       0
Bank Sta=311,332.9
XS Rating Curve= 0 ,0
Exp/Cntr(USF)=0,0
Exp/Cntr=0.3,0.1

Type RM Length L Ch R = 1 ,16577   ,587.1,592.8,581.6
XS GIS Cut Line= 3
 1655808.4036836430864.7570908551655976.61918578430729.617145603
1656144.67969838430350.664295933
#Sta/Elev= 30
       0 1163.39    14.2 1158.92    48.3    1145    76.8 1137.05   122.3 1121.08
   148.4 1113.74   172.8 1105.38   179.2 1101.48   190.6 1090.49   204.8  1078.8
   211.1 1075.09   221.3 1073.66   260.7 1074.38   276.8 1073.32   281.8 1074.33
     287 1075.72   304.5 1077.49   316.2 1080.54   348.2 1094.55   373.8 1104.41
   401.1 1113.14   431.4 1127.78   453.2 1128.35   466.4 1136.05   483.9  1142.9
     497 1150.97   570.9 1189.26   597.6 1204.53   607.3 1208.23   630.3 1218.99
#Mann= 5 ,-1,0
       0      .1       0   260.7    .045       0   281.8      .1       0
  335.78     .06       0  445.78      .1       0
Bank Sta=260.7,281.8
XS Rating Curve= 0 ,0
Exp/Cntr(USF)=0,0
Exp/Cntr=0.3,0.1

Type RM Length L Ch R = 1 ,15985   ,413.7,412.5,409.2
BEGIN DESCRIPTION:
Structure XS 4
END DESCRIPTION:
XS GIS Cut Line= 6
1656457.49928884431097.5167118461656458.91890542431001.277403012
1656452.66629326430911.7841436711656398.20511609430741.152595177
1656386.62803951430661.1583325861656385.73040351430469.563899502
#Sta/Elev= 30
       0 1147.49      21 1140.21      41 1135.87    82.4 1131.82     105 1127.29
   145.8 1113.02   169.2 1101.92   185.2    1097   231.2 1072.54   247.9 1070.51
   297.5 1069.28   303.9 1068.08     311 1066.71   319.4 1068.04   344.7 1067.89
   348.9 1069.11   360.9 1076.54     394  1091.2   402.1  1095.9   414.2 1105.14
   422.3 1106.52   438.5 1106.75   450.5 1114.17   454.5 1115.41   466.5 1125.05
   482.5 1129.97   498.6 1131.77   554.4 1161.44   594.6 1180.31   637.6 1203.44
#Mann= 5 ,-1,0
       0      .1       0   303.9    .045       0   319.4      .1       0
  395.08     .06       0  485.91      .1       0
Bank Sta=303.9,319.4
XS Rating Curve= 0 ,0
Exp/Cntr(USF)=0,0
Exp/Cntr=0.3,0.1

Type RM Length L Ch R = 1 ,15572   ,40,41.1,42.2
BEGIN DESCRIPTION:
Structure XS 3
END DESCRIPTION:
XS GIS Cut Line= 6
1656728.57665154431092.2874161381656793.29611223430941.275341195
1656815.69900247430860.7908836711656791.63663888430809.347209789
1656762.59585523430796.0714229811656682.94113438 430533.87463352
#Sta/Elev= 30
       0 1137.21    51.2 1122.89    86.8 1114.86   104.2    1109   120.7 1101.22
     141 1089.77   147.7 1084.68   160.7  1072.1   165.1  1069.7   185.8 1066.54
     274 1065.88   278.7  1063.9   292.2 1062.41   298.2 1063.86   308.8 1068.19
   316.5 1072.62   326.2    1075   335.8 1076.43   377.9 1078.34   386.2 1084.17
   390.4 1085.97     407 1087.67   419.7 1090.86   465.6 1108.81     495 1118.72
   511.7 1126.88   550.5  1141.7   588.8  1162.3     604 1166.25     611 1169.96
#Mann= 6 ,-1,0
       0      .1       0   194.3     .05       0   278.7    .045       0
   298.2     .05       0  301.52     .06       0   524.4      .1       0
Bank Sta=278.7,298.2
XS Rating Curve= 0 ,0
Exp/Cntr(USF)=0,0
Exp/Cntr=0.3,0.1

Type RM Length L Ch R = 1 ,15531   ,194.3,210.3,221.3
BEGIN DESCRIPTION:
Structure XS 2
END DESCRIPTION:
XS GIS Cut Line= 6
1656742.68217502431100.5847828931656848.05873281430878.215353857
1656847.22899613430843.366413485 1656831.4639993 430801.87957971
1656813.20979244430784.4551095241656725.25770483430528.066476792
#Sta/Elev= 30
       0 1136.33    17.8  1132.1    52.2 1121.99    79.7 1116.81   112.3 1106.69
   145.3 1089.85   150.5 1084.56   154.9 1077.95   157.3 1075.86   168.2 1068.93
   172.6 1067.18   190.3 1065.53     284 1065.01   289.7 1063.61     301 1061.81
   309.6 1063.64   318.2 1067.96   338.8 1072.72   371.8 1074.29   380.3 1076.83
   397.4 1079.53   405.9 1083.53   461.4 1101.03   482.7 1109.58   512.6 1119.75
   533.9 1129.73   563.4 1139.26   579.8 1146.25   596.6 1154.86   621.9 1165.01
#Mann= 7 ,-1,0
       0      .1       0  190.73     .06       0  210.73     .05       0
   289.7    .045       0   309.6     .05       0  310.93     .06       0
  530.55      .1       0
Bank Sta=289.7,309.6
XS Rating Curve= 0 ,0
Exp/Cntr(USF)=0,0
Exp/Cntr=0.3,0.1

Type RM Length L Ch R = 1 ,15321   ,433.3,434.7,433.3
BEGIN DESCRIPTION:
Structure XS 1
END DESCRIPTION:
XS GIS Cut Line= 3
1656751.93334163431118.2474465521656873.78056975 430997.69743513
1657275.67042021430747.066211496
#Sta/Elev= 30
       0 1137.83   101.5 1106.11   129.7 1093.08   165.4 1067.04   173.9 1063.67
   221.3 1062.27   287.3 1063.22   339.1 1061.75     351 1059.88   356.9 1060.47
   359.8 1061.87   362.7 1064.05   367.4    1070   372.1 1073.56   377.7 1074.69
   391.7 1075.06   395.7 1077.14   409.9 1088.71   414.6 1090.33   428.7 1091.33
   438.1 1096.81   449.8 1102.11   483.5 1113.33     523 1130.03   542.7 1136.23
     556 1141.86   598.4 1166.38   618.2 1172.39   632.7 1178.49     645 1180.91
#Mann= 7 ,-1,0
       0      .1       0     150     .06       0   231.4      .1       0
   331.4     .06       0   339.1    .045       0   359.8     .06       0
   461.4      .1       0
Bank Sta=339.1,359.8
XS Rating Curve= 0 ,0
Exp/Cntr(USF)=0,0
Exp/Cntr=0.3,0.1

Type RM Length L Ch R = 1 ,14886   ,330.1,330.8,330
BEGIN DESCRIPTION:
Structure XS 4
END DESCRIPTION:
XS GIS Cut Line= 2
1656957.41203302431453.1292784391657440.18940582431117.650821729
#Sta/Elev= 30
       0 1150.26    22.8 1142.23    50.1 1135.72    74.2 1127.68   110.5 1117.74
   148.2    1104   183.4 1088.92     203 1076.32   212.7 1068.82   232.2 1059.14
   258.1 1056.99   263.9 1055.73   263.9 1055.72   271.2 1054.09   280.9 1055.74
   341.5 1058.47   367.4 1057.71   379.6 1059.83   387.5 1063.98   401.8 1078.29
   407.5 1083.12   412.4 1085.86   427.1 1087.39   441.7 1097.86   453.6 1102.92
   467.9 1111.71   496.7  1121.4     534 1136.47   561.8 1145.71   587.9 1157.82
#Mann= 5 ,-1,0
       0      .1       0   263.9    .045       0   280.9      .1       0
     320     .06       0     440      .1       0
Bank Sta=263.9,280.9
XS Rating Curve= 0 ,0
Exp/Cntr(USF)=0,0
Exp/Cntr=0.3,0.1

Type RM Length L Ch R = 1 ,14555   ,63.4,63.4,63.6
BEGIN DESCRIPTION:
Structure XS 3
END DESCRIPTION:
XS GIS Cut Line= 5
1657312.66007248431735.1442223221657392.64579288 431533.78373897
 1657470.0409793431470.4590624561657521.54907838431408.000745734
1657625.44599148431253.211496405
#Sta/Elev= 30
       0 1155.11    72.4 1139.02    93.2  1132.3   114.7 1123.25   136.2 1116.64
   153.4 1108.04   180.3 1089.13   192.2 1078.71   200.8 1067.83     208  1063.1
   211.1 1062.27   243.9 1061.28   252.2 1058.71   262.9 1051.66   268.3 1049.92
   272.8 1049.62   285.4 1051.55   314.2 1054.83   338.8 1060.68   376.2 1062.73
   391.7 1073.05   399.1 1077.02   433.7 1090.38   445.2 1092.15     450 1094.34
   459.6 1100.73   474.1 1105.85   538.6 1134.91   551.9 1138.32     584 1153.77
#Mann= 5 ,-1,0
       0     .05       0     140      .1       0   262.9    .045       0
   285.4     .06       0  396.67      .1       0
Bank Sta=262.9,285.4
XS Rating Curve= 0 ,0
Exp/Cntr(USF)=0,0
Exp/Cntr=0.3,0.1

Type RM Length L Ch R = 1 ,14492   ,500,500,496.2
BEGIN DESCRIPTION:
Structure XS 2
END DESCRIPTION:
XS GIS Cut Line= 5
1657361.13167994431777.1072098651657441.11740033431575.746726513
1657518.51258676431512.4220499991657570.02068584431449.963733278
1657673.91759893431295.174483949
#Sta/Elev= 30
       0 1168.89    61.3 1148.29    95.3 1137.88   112.5 1131.34     129 1123.81
     147 1117.85   172.8 1102.06   181.4 1095.12     190  1086.1   207.2 1070.14
   221.7 1058.85   228.1 1056.37   246.7 1053.66  255.67 1051.01   263.7 1049.32
   275.1 1049.74   280.8 1050.97   287.7 1052.11   320.6 1054.01   337.6 1058.41
   383.1 1060.12   397.6 1070.23     403 1073.05   446.3 1088.46   460.7  1091.2
   476.4 1101.07   523.4 1120.66   535.6 1123.54   550.1 1131.24     584 1143.95
#Mann= 6 ,-1,0
       0     .05       0     190      .1       0  255.67    .045       0
   280.8      .1       0  326.67     .06       0  447.62      .1       0
Bank Sta=255.67,280.8
XS Rating Curve= 0 ,0
Exp/Cntr(USF)=0,0
Exp/Cntr=0.3,0.1

Type RM Length L Ch R = 1 ,13992   ,409.3,409.1,407.3
BEGIN DESCRIPTION:
Structure XS 1
END DESCRIPTION:
XS GIS Cut Line= 6
1657719.56533426431930.9425384251657774.13641934431851.902998343
1657836.48504792431790.4880949261657890.93113326431738.906833261
1657963.52711667431670.1333487631658149.55200709431493.898136929
#Sta/Elev= 30
       0 1146.36    13.6 1141.09    71.1 1114.59   102.7  1101.7   117.9 1092.89
   139.4 1088.18   194.1 1065.06   227.1 1049.78   232.8 1047.94   250.4 1046.57
   286.5 1046.22   293.3 1044.62   297.9 1042.46   302.7 1040.47   306.3 1040.21
   315.3 1040.49  319.811042.439   332.2 1049.52   343.1 1058.02   374.3 1088.86
   378.3 1090.47   392.4 1091.19   403.5 1100.53   425.5 1114.39     442 1121.74
   476.1 1134.87   488.8 1138.89   529.6 1148.44   589.3 1172.26   614.8 1178.69
#Mann= 5 ,-1,0
       0     .05       0  288.56      .1       0   297.9    .045       0
  319.81     .06       0  453.56      .1       0
Bank Sta=297.9,319.81
XS Rating Curve= 0 ,0
Exp/Cntr(USF)=0,0
Exp/Cntr=0.3,0.1

Type RM Length L Ch R = 1 ,13583   ,138.5,136.6,132.6
BEGIN DESCRIPTION:
Structure XS 4
END DESCRIPTION:
XS GIS Cut Line= 6
1657963.17566011432248.1239217511658087.72856062432116.449644415
1658207.98685029431989.316040425 1658259.5257892431934.829928918
1658319.09194303431870.730647667 1658382.6062517431801.719302757
#Sta/Elev= 30
       0 1147.68      13 1144.68    53.8 1129.54   123.6 1098.67   148.1  1089.7
   164.5 1082.31   187.6 1070.51   212.6  1051.6   226.7 1044.21   235.2 1042.68
   274.8 1042.34   294.6 1038.73   302.3 1035.61   307.8 1035.29   313.3 1035.75
   320.1 1038.68   334.3 1043.19   351.2 1057.54   368.1 1059.12   373.9 1065.82
   379.5 1070.62   396.5 1071.33   407.8 1080.53   441.8 1094.55   450.8 1097.07
   494.4 1122.76   512.5 1129.11     538 1141.22   581.5 1153.82   612.5 1174.17
#Mann= 5 ,-1,0
       0      .1       0      70     .05       0   294.6    .045       0
   320.1     .05       0  346.25      .1       0
Bank Sta=294.6,320.1
XS Rating Curve= 0 ,0
Exp/Cntr(USF)=0,0
Exp/Cntr=0.3,0.1

Type RM Length L Ch R = 1 ,13446   ,54,52.5,52.8
BEGIN DESCRIPTION:
Structure XS 3
END DESCRIPTION:
XS GIS Cut Line= 3
1658199.31626518432406.187535897 1658201.3325253432258.328460321
1658423.12113867431830.881314566
#Sta/Elev= 30
       0 1110.62    13.7 1105.83    41.7 1093.03    57.7 1088.94    73.7  1083.1
    85.7 1074.61    97.1 1068.06   137.7 1049.85   226.5 1044.41     258 1040.66
   290.7  1039.6     3001036.106   303.1 1034.58   312.1    1034   320.4 1036.11
   329.3 1041.48   343.7 1042.23   347.1 1043.59   357.2 1052.21   375.2  1063.3
   382.7 1065.04   411.3 1066.83   442.8 1080.79   465.8 1089.39   492.5 1102.45
   557.7 1139.14     567 1142.97   600.5 1152.93   613.9 1160.16   629.4 1170.88
#Mann= 8 ,-1,0
       0      .1       0      20     .05       0     120     .06       0
  217.87     .05       0     300    .045       0   320.4     .05       0
  327.87     .06       0  447.87      .1       0
Bank Sta=300,320.4
XS Rating Curve= 0 ,0
Exp/Cntr(USF)=0,0
Exp/Cntr=0.3,0.1

Type RM Length L Ch R = 1 ,13394   ,403.9,401.7,399.8
BEGIN DESCRIPTION:
Structure XS 2
END DESCRIPTION:
XS GIS Cut Line= 3
1658241.65772773432404.1712757751658244.34607456432291.260708972
 1658464.1184278 431853.73226261
#Sta/Elev= 30
       0 1110.21    47.6 1086.99    63.7  1081.5    71.7 1075.42   111.7 1049.64
   124.9 1047.34   162.5  1044.2   248.9 1039.54  258.211035.495   268.2 1033.55
   281.7 1035.41   281.7 1035.43   293.6  1037.2   299.5 1039.28   312.9 1051.85
   326.4 1060.85   335.3 1064.82   356.1  1066.2   366.7 1072.49   379.8  1074.6
   388.7 1077.23   411.4 1086.99   442.6  1096.1   487.2 1118.29   514.4  1130.2
   532.3 1139.66   541.2 1143.16   573.7 1151.72   590.5 1158.75   602.6 1165.99
#Mann= 9 ,-1,0
       0      .1       0      10     .05       0     110     .06       0
  222.94     .05       0  242.94     .08       0  258.21    .045       0
   281.7     .08       0  332.94     .06       0  442.94      .1       0
Bank Sta=258.21,281.7
XS Rating Curve= 0 ,0
Exp/Cntr(USF)=0,0
Exp/Cntr=0.3,0.1

Type RM Length L Ch R = 1 ,12992   ,488.5,499.9,506.6
BEGIN DESCRIPTION:
Structure XS 1
END DESCRIPTION:
XS GIS Cut Line= 6
1658585.61707984432631.5625282531658619.95264108 432543.48101151
1658639.55693258  432458.20559151658656.36004859432385.111905679
1658715.17095459432129.2846614271658737.62399368432038.251050845
#Sta/Elev= 30
       0 1135.91    20.4 1122.78    50.5 1105.33   105.8 1075.35   130.4 1063.37
   146.8 1049.15   167.3 1035.39   175.5 1033.91   290.5 1034.17  296.941032.813
   302.8 1031.72     311 1031.88   315.1  1032.8   335.6 1035.84   343.8 1038.95
   350.8 1043.92   368.4 1059.23   372.5 1061.13   384.9 1062.19     389  1064.9
   400.8 1075.25   413.6 1083.16   495.7 1124.86   512.1 1130.32   528.5 1138.73
     545 1145.13   565.6 1151.61   582.1 1155.63   594.5 1160.21   613.3 1169.68
#Mann= 6 ,-1,0
       0      .1       0  154.54     .05       0  252.04     .06       0
  296.94    .045       0   315.1     .06       0  427.04      .1       0
Bank Sta=296.94,315.1
XS Rating Curve= 0 ,0
Exp/Cntr(USF)=0,0
Exp/Cntr=0.3,0.1

Type RM Length L Ch R = 1 ,12492   ,499.1,500.1,498.1
XS GIS Cut Line= 6
1658719.99246725432744.5104650861658816.08709134432704.321569085
1658908.05508326 432677.343276591658985.05525734432657.381702334
1659149.07986367432596.3486879171659317.28950101432528.545673922
#Sta/Elev= 30
       0 1131.46    30.5 1120.14    65.2 1104.66    82.9 1095.04     104 1079.32
   129.8  1077.5   141.7 1074.19   154.2 1065.33   175.1 1047.49   204.2 1030.98
     227 1027.79   243.4 1029.41   266.2  1028.4   287.1 1031.26   310.7 1030.86
  318.991028.675   329.6 1027.09   336.6 1028.63   351.3 1037.92   364.2 1042.01
   367.9 1044.98   376.4 1055.76   402.1 1079.29     415 1080.76   419.6 1083.62
   427.8 1092.72     432 1095.67   487.9 1119.91   542.1 1134.91   635.9 1151.74
#Mann= 7 ,-1,0
       0      .1       0  184.16     .05       0  289.55      .1       0
  318.99    .045       0   336.6      .1       0  389.55     .06       0
  494.57      .1       0
Bank Sta=318.99,336.6
XS Rating Curve= 0 ,0
Exp/Cntr(USF)=0,0
Exp/Cntr=0.3,0.1

Type RM Length L Ch R = 1 ,11992   ,491.1,500,504.4
XS GIS Cut Line= 6
1658900.88941517433208.4015976791659067.22668092433136.405678675
1659227.82839385433066.8920381671659296.63665517433037.051546678
1659376.75657368433001.8774044221659462.53264885432964.036600843
#Sta/Elev= 30
       0 1147.48    60.3 1113.99    68.9 1108.14    86.3 1100.79    99.7 1092.57
   130.6  1076.3   139.2 1069.89   151.4 1054.54   160.4 1047.05   177.9 1043.54
     191 1031.94   200.1 1025.72   208.4 1023.88   269.4    1023   294.4 1021.47
   303.5  1019.8     313 1020.09  316.681021.529   327.8 1034.37   339.1 1040.93
   370.4 1051.62   382.7 1058.71   400.2 1066.42   448.2 1084.22   496.2 1104.08
   513.7 1112.28   526.8 1120.42   535.5 1123.14     553 1131.82   612.5 1153.14
#Mann= 3 ,-1,0
       0      .1       0   294.4    .045       0  316.68      .1       0
Bank Sta=294.4,316.68
XS Rating Curve= 0 ,0
Exp/Cntr(USF)=0,0
Exp/Cntr=0.3,0.1

Type RM Length L Ch R = 1 ,11492   ,511.7,500,491.3
XS GIS Cut Line= 6
1659002.86198026433527.2310125081659096.32111092433534.609606668
1659258.31717801433547.3976388421659358.00693926433555.267701834
1659520.00300634433568.0547497571659613.74035168433571.909400836
#Sta/Elev= 30
       0 1094.32    29.3 1074.83    65.6 1057.69    81.5 1056.29    97.6 1050.77
   129.7 1045.52   149.7 1040.18   165.8 1039.56   169.8 1038.48   197.9 1026.49
   205.9 1024.04     242 1019.98   282.1 1018.12   290.2 1016.29   298.2 1015.01
   317.61016.298   342.3 1019.33   346.3 1021.48   350.3 1024.99   358.4 1036.61
   362.4 1040.21   386.5  1051.7   402.5 1063.91   418.6 1072.54   438.6 1078.68
   458.7 1087.85   546.2 1134.41   568.5 1142.42   594.9 1154.11   612.6 1160.44
#Mann= 3 ,-1,0
       0      .1       0   290.2    .045       0   317.6      .1       0
Bank Sta=290.2,317.6
XS Rating Curve= 0 ,0
Exp/Cntr(USF)=0,0
Exp/Cntr=0.3,0.1

Type RM Length L Ch R = 1 ,10992   ,487,500,506.4
XS GIS Cut Line= 6
1659228.75555734434111.6474945841659410.58130917434045.822823092
1659483.04310651 434014.417046011659616.38109443433901.076721504
1659682.43181534433843.6910095071659751.38935459433779.973289177
#Sta/Elev= 30
       0 1142.39    16.3 1130.93    33.4 1114.73    42.5 1107.51    46.2 1103.56
      54 1092.49    67.4 1076.26    79.9 1065.69      93 1057.39   105.8  1054.2
   139.8 1041.84   186.5 1040.37   203.8 1038.09   234.3 1025.24   253.3 1014.48
   259.4 1012.37     300 1012.84   308.5 1011.99     317 1010.52   331.5 1011.98
   342.5 1014.01   386.4 1016.86   429.7 1024.06   453.2  1033.5   473.5  1037.8
     500 1045.65   518.4 1054.52   563.1  1083.9   592.1 1095.27   628.7 1115.35
#Mann= 3 ,-1,0
       0      .1       0   308.5    .045       0   331.5      .1       0
Bank Sta=308.5,331.5
XS Rating Curve= 0 ,0
Exp/Cntr(USF)=0,0
Exp/Cntr=0.3,0.1

Type RM Length L Ch R = 1 ,10492   ,517.5,501.9,492.3
XS GIS Cut Line= 6
1659236.35003035434426.920814171 1659329.5316025 434437.27873309
1659590.71972843434463.4902948441659665.17561626434472.673675418
1659751.98777859434483.9151227621659846.03319417434489.518129915
#Sta/Elev= 30
       0 1024.73    48.1 1021.15    84.6  1023.6   100.4 1023.17   108.4 1021.98
   124.5 1018.43   180.8 1015.65   208.9 1012.27   269.2 1009.04   281.8 1007.85
  292.07 1005.32   297.4 1004.55   309.4 1004.67   313.4 1005.25   321.5 1007.16
   325.5 1009.16   333.5 1016.42   341.6 1021.66   349.6 1025.61   373.8 1033.06
   393.9 1040.49   434.2 1052.12   446.3 1054.99   462.3 1060.81   486.7 1072.71
   506.8 1080.95     571 1105.45   595.2 1113.16   599.1 1114.93     613  1123.4
#Mann= 3 ,-1,0
       0      .1       0  292.07    .045       0   313.4      .1       0
Bank Sta=292.07,313.4
XS Rating Curve= 0 ,0
Exp/Cntr(USF)=0,0
Exp/Cntr=0.3,0.1

Type RM Length L Ch R = 1 ,9990    ,487.4,497,502.2
XS GIS Cut Line= 6
1659570.13020268435111.1002200841659718.63515501434902.269601002
1659779.81154184434823.0666754251659829.03978984434765.640281096
1659886.22110592434698.2509801691659947.84106143434626.662540674
#Sta/Elev= 30
       0  1141.9    17.9 1131.55    31.9  1120.4    57.1  1108.1    80.7 1092.01
   100.8 1082.81   120.8 1065.84   135.7 1056.59     170 1040.85   189.7 1036.18
   204.4 1027.89   218.4 1023.96   238.5 1022.03   253.5 1017.57   278.3 1006.71
   287.1 1000.85   297.9  998.83   318.4  1000.8   329.2 1002.22   352.6  1002.4
   359.7 1004.22   389.5 1022.77   409.4 1033.46   420.7 1044.01   426.4 1047.95
   455.3 1058.51     486 1078.42   539.9 1107.03   591.2 1138.18   614.8  1149.5
#Mann= 3 ,-1,0
       0      .1       0   287.1    .045       0   318.4      .1       0
Bank Sta=287.1,318.4
XS Rating Curve= 0 ,0
Exp/Cntr(USF)=0,0
Exp/Cntr=0.3,0.1

Type RM Length L Ch R = 1 ,9493    ,493.8,493.8,487.2
XS GIS Cut Line= 6
1659744.50157309435401.964467749  1659972.666143435273.821679428
1660065.86805634435233.7728750111660135.81115793435206.699766427
  1660203.224737 435147.046998591660264.68885292435069.446103916
#Sta/Elev= 30
       0 1126.28    91.5 1093.36   121.1 1078.43   132.8 1069.11   146.6 1063.74
   165.6  1054.5     171 1050.53   181.9 1039.53     197 1030.94   212.2 1027.49
     221 1021.25   238.2 1011.34   247.5 1009.29   261.1 1003.54   277.5  1001.7
   286.6  996.68  293.32994.6518   298.8  994.11     314  994.64   326.2   996.6
   356.6 1011.39   374.1 1018.46   445.5 1036.16   486.6 1053.15     524 1064.65
   548.9 1078.54   582.4 1093.34   606.9 1108.11   618.1 1111.34   627.1 1118.01
#Mann= 3 ,-1,0
       0      .1       0  293.32    .045       0     314      .1       0
Bank Sta=293.32,314
XS Rating Curve= 0 ,0
Exp/Cntr(USF)=0,0
Exp/Cntr=0.3,0.1

Type RM Length L Ch R = 1 ,8999    ,484.2,499.1,500.4
XS GIS Cut Line= 6
1660164.92166401435730.170504257 1660234.2564991435660.076156259
1660345.28121142435541.534070507 1660412.0238601435465.631991342
1660462.41385117435405.7859824151660584.25087784435264.142564923
#Sta/Elev= 30
       0 1114.42    20.4 1108.76    37.4 1099.93      50 1096.18    91.1 1069.29
   119.4 1056.94   136.4 1043.85   152.8 1038.74   169.2  1029.4   178.8 1027.17
   190.1 1018.91   207.1 1011.05   224.2  998.92   235.4  993.15   259.3  991.17
   292.1  992.07   307.7  988.57   311.9  988.22   334.6  988.52   347.6  994.68
   368.7 1020.29   377.1 1027.81   408.3 1037.92   436.7 1057.66   448.1 1059.13
   468.3 1066.15   489.4 1081.29     570 1129.09   608.5 1147.07   627.2 1152.96
#Mann= 3 ,-1,0
       0      .1       0   307.7    .045       0   334.6      .1       0
Bank Sta=307.7,334.6
XS Rating Curve= 0 ,0
Exp/Cntr(USF)=0,0
Exp/Cntr=0.3,0.1

Type RM Length L Ch R = 1 ,8500    ,494.4,498.2,495.2
XS GIS Cut Line= 6
1660396.39561051436010.3287365881660564.05898909435878.357543841
1660642.65922558435818.2746587541660805.50798126435754.201296091
1660887.04882868435722.4615301791660974.57457225435688.862187922
#Sta/Elev= 30
       0  1042.1    48.1 1037.06     115 1021.56   137.2 1014.19   169.1  996.32
   183.4  995.72   198.2   990.9   246.1  989.28   277.5  986.38   313.9  986.25
   335.4  984.95     344  982.82   361.2  981.78  378.85982.9484   415.4 1007.99
   429.9 1021.35   438.5 1035.38   442.8 1039.88   455.7 1045.95   477.2 1059.69
   499.9  1068.1   515.9 1076.27     540 1090.97   558.6  1099.8   570.9 1103.21
   601.1 1122.33     636 1137.65   648.3 1144.43   658.3 1146.88   668.6 1153.25
#Mann= 3 ,-1,0
       0      .1       0     344    .045       0  378.85      .1       0
Bank Sta=344,378.85
XS Rating Curve= 0 ,0
Exp/Cntr(USF)=0,0
Exp/Cntr=0.3,0.1

Type RM Length L Ch R = 1 ,8002    ,508.6,502,494.4
XS GIS Cut Line= 6
1660623.10873976436323.395039588 1660779.5231251436220.624903917
1660850.65159176436195.9953600021660948.54575293436175.255900174
  1661018.345154436140.8356934191661175.21787176436027.640381753
#Sta/Elev= 30
       0 1156.97    57.3 1118.13    65.9 1110.75    94.7 1093.53   117.9 1076.63
   135.4 1066.28     147 1064.63   164.5 1050.76   178.6 1043.77   196.3 1025.21
   209.8 1015.72   228.7  997.32   238.7  992.17   251.4  989.39   266.7  983.17
  299.99977.2465   321.3   977.2   337.1  976.63   370.3  979.29   384.4  984.85
   404.9 1000.14   415.1 1013.03   441.9 1037.53   464.9 1047.35   483.4  1061.1
   519.6  1075.3   559.8 1101.29   572.7 1105.34   584.9 1114.04   633.9 1141.35
#Mann= 3 ,-1,0
       0      .1       0  299.99    .045       0   321.3      .1       0
Bank Sta=299.99,321.3
XS Rating Curve= 0 ,0
Exp/Cntr(USF)=0,0
Exp/Cntr=0.3,0.1

Type RM Length L Ch R = 1 ,7500    ,481.9,497.3,500.1
XS GIS Cut Line= 6
1661016.92192851436782.6349347531661132.41283926436642.705096513
1661180.75690268436585.3046207581661247.59010234436510.917958513
1661356.56757468436390.3768610061661418.51692584436320.000033259
#Sta/Elev= 30
       0 1163.18    57.8 1128.32      96 1102.97   111.7 1095.71   140.1  1074.6
   162.2 1067.75   179.9 1054.72     200 1044.11   228.2 1019.51   239.5 1004.52
   259.4  988.24   273.6   984.2  297.19  971.89   316.7  971.09   324.5  971.91
   341.5  974.93   386.7  974.87   397.4   978.8     405  983.96   415.2   993.8
   435.2 1017.37   467.5  1041.2   494.5 1054.36   508.6 1064.79   537.4 1075.96
   548.6 1082.77   565.3 1096.53   580.1 1100.77     603 1116.67   612.7  1121.3
#Mann= 3 ,-1,0
       0      .1       0  297.19    .045       0   324.5      .1       0
Bank Sta=297.19,324.5
XS Rating Curve= 0 ,0
Exp/Cntr(USF)=0,0
Exp/Cntr=0.3,0.1

Type RM Length L Ch R = 1 ,7003    ,487.7,498.4,505.3
XS GIS Cut Line= 6
1661201.71486601436944.3957660941661289.44959867436908.512963846
1661374.90316792436889.209196672  1661622.623473436839.042302251
  1661713.505181436831.6082620021661810.31141783436828.009187832
#Sta/Elev= 30
       0  1118.7    32.8 1099.01    50.1 1083.48      63 1075.85    94.8 1068.46
     118 1056.45   142.6 1048.46   187.7 1017.86   212.2  995.08   240.8  974.22
     249  970.95   282.1  970.07   289.8  968.02     298  966.66     316  968.11
   351.1  969.87   371.5  967.35   383.7  968.41   391.8  975.69   424.9  991.04
   444.7 1004.61   472.8 1029.23   488.8 1045.41   500.9 1051.47   516.9 1065.21
     537 1072.84     585 1107.94   593.6 1110.93   604.8 1119.61   623.2 1130.33
#Mann= 3 ,-1,0
       0      .1       0   289.8    .045       0     316      .1       0
Bank Sta=289.8,316
XS Rating Curve= 0 ,0
Exp/Cntr(USF)=0,0
Exp/Cntr=0.3,0.1

Type RM Length L Ch R = 1 ,6504    ,503.1,505.5,491.7
XS GIS Cut Line= 6
1661158.12735476437161.1518942561661372.97535026  437300.8100795
1661464.66808026437350.2007287591661553.49861126437363.730885416
1661658.51480542437359.8821398321661768.91550326437335.703382418
#Sta/Elev= 30
       0 1066.22     7.1 1063.96    20.9 1055.41    29.9 1051.23    78.7 1038.79
     109 1027.83   131.2 1015.84   169.3  985.66   188.4  976.72   211.7  973.21
   221.8   973.7   287.1  967.52   296.2  962.96   300.7  962.27  321.63962.9672
   346.1   965.2     372   964.3   416.5  965.61   436.7   975.6   444.8  980.65
   460.9  993.14   480.9 1012.07   516.9  1033.6   544.9 1047.21   565.2 1053.14
   577.5 1061.29   597.9 1067.03   630.7 1081.81   651.2 1094.98   668.4  1101.5
#Mann= 3 ,-1,0
       0      .1       0   296.2    .045       0  321.63      .1       0
Bank Sta=296.2,321.63
XS Rating Curve= 0 ,0
Exp/Cntr(USF)=0,0
Exp/Cntr=0.3,0.1

Type RM Length L Ch R = 1 ,5999    ,487.5,498.7,505.3
XS GIS Cut Line= 6
1661364.06821585437846.5990141781661456.69073401437795.807121009
1661547.05636692437747.0522972491661624.29144867437706.623572335
1661724.22628817437702.1239094291661980.43476526437697.509089261
#Sta/Elev= 30
       0 1102.15    54.8 1072.81      73 1068.56    95.9 1055.97   118.6 1047.06
   123.2 1043.13     143 1019.27   163.7  1000.5   181.4   986.7   216.9  965.85
   232.1  962.61   319.3  960.45   326.8958.5787   335.6   957.5   355.4  958.53
   371.4  969.32   383.4  970.32   403.4  974.85   455.4 1000.17   499.2 1024.87
   523.4 1045.08   531.4 1048.47   539.4  1049.1   546.3  1051.6   555.4 1059.78
   563.4 1064.66   603.4 1077.54   624.9 1093.77   639.5 1099.98   651.8 1107.26
#Mann= 3 ,-1,0
       0      .1       0   326.8    .045       0   355.4      .1       0
Bank Sta=326.8,355.4
XS Rating Curve= 0 ,0
Exp/Cntr(USF)=0,0
Exp/Cntr=0.3,0.1

Type RM Length L Ch R = 1 ,5500    ,510,500.1,492.5
XS GIS Cut Line= 6
1661399.03304093438018.2541826671661496.38323992438037.937214166
1661577.93983534438073.9850423341661640.46136384438115.421639249
 1661723.0842301438171.7555160821661934.80395101438316.112182751
#Sta/Elev= 30
       0 1070.17    17.4  1065.8    29.7  1060.1    41.9 1051.78    58.2 1047.21
    82.7 1028.96    90.9 1021.02   104.1 1018.19   116.5 1010.68   125.3  1007.9
   138.4 1006.44   147.1 1002.88     169  998.04   200.3  985.42   229.5  978.46
   281.3  956.24   292.1  953.11   301.5   952.9   315.2  951.98   327.4     953
     336  961.18   367.7  981.17   400.4  991.35   433.9    1007   448.3 1011.31
   519.7 1045.96   534.2 1050.73   563.2 1056.89   592.2 1068.66   619.7  1074.1
#Mann= 3 ,-1,0
       0      .1       0   301.5    .045       0   327.4      .1       0
Bank Sta=301.5,327.4
XS Rating Curve= 0 ,0
Exp/Cntr(USF)=0,0
Exp/Cntr=0.3,0.1

Type RM Length L Ch R = 1 ,5000    ,496.4,493.9,489.8
XS GIS Cut Line= 6
1661303.83670901438747.7146660091661535.30146918438637.768691674
1661625.77799426438595.0722547621661697.45468818438567.597900257
 1661784.6290545438541.5940152561661878.77158275438512.636724085
#Sta/Elev= 30
       0 1043.07    26.9 1040.53    84.4 1028.22    93.3 1026.95   150.9 1013.95
   168.6 1011.07     204 1002.71   251.8  985.62     266  979.03   270.4  976.33
   275.8  971.05   279.3  966.11   284.8  955.78   288.1  951.11  296.67  947.57
   301.4  946.77   308.9  947.58   323.5  950.38   363.2  951.23   375.9  955.94
   387.9  956.77   405.9  959.93   414.5  962.65     440   972.9   460.9  979.26
   530.9  989.87   543.7  994.43   565.3 1005.88   577.9 1011.09   622.5 1035.02
#Mann= 3 ,-1,0
       0      .1       0  296.67    .045       0   308.9      .1       0
Bank Sta=296.67,308.9
XS Rating Curve= 0 ,0
Exp/Cntr(USF)=0,0
Exp/Cntr=0.3,0.1

Type RM Length L Ch R = 1 ,4506    ,504.3,505.8,490.9
XS GIS Cut Line= 6
1661708.68334025439231.1897489281661805.97284384439076.000426754
1661920.88534367438941.0620483461661948.64020942438864.665219501
1661972.14541176438774.504310593 1662009.8923835438679.036981836
#Sta/Elev= 30
       0 1152.84    40.4 1126.56    54.4 1114.19    63.7  1111.8    68.4 1109.14
    80.2 1099.07    91.7 1092.21   101.2 1078.74   123.7 1070.61   128.9 1067.25
     141  1051.4   158.4 1042.53     193 1008.86   213.3  993.55     227  979.54
     263  958.22   299.1  941.54   309.3  940.94   323.7  941.52   350.5  944.12
   361.1  948.31   369.6  948.37   382.3  952.07   399.4  952.43   462.6  976.32
   491.5  988.96   532.9 1002.07   562.9 1006.69   614.5 1020.07   637.6 1030.25
#Mann= 3 ,-1,0
       0      .1       0   299.1    .045       0   323.7      .1       0
Bank Sta=299.1,323.7
XS Rating Curve= 0 ,0
Exp/Cntr(USF)=0,0
Exp/Cntr=0.3,0.1

Type RM Length L Ch R = 1 ,4000    ,471.1,500.1,514.4
XS GIS Cut Line= 6
1662256.71144368439358.7547825131662309.19591875439272.932775676
1662327.54168259439187.3512539271662342.93633685 439113.93374984
1662361.72435701439015.7141299991662409.36041659438763.930840924
#Sta/Elev= 30
       0 1078.12    14.2  1074.5    35.4 1060.91    68.2 1049.25    82.3  1042.6
   133.7 1007.16     146  996.33   158.3  992.01   182.8  973.74   223.7  949.59
   251.8  943.42   268.6  943.63   280.9   938.4  295.24934.7507   309.4  934.06
   325.6  934.74   337.9  935.29   354.2  939.94   390.8  944.67   411.2  951.03
   423.4  959.74   447.8   981.4   500.7 1016.81     517 1029.41   534.8 1048.58
   557.7 1070.26   590.3 1075.95   598.4 1080.77   607.5 1089.93   619.4 1097.26
#Mann= 3 ,-1,0
       0      .1       0  295.24    .045       0   325.6      .1       0
Bank Sta=295.24,325.6
XS Rating Curve= 0 ,0
Exp/Cntr(USF)=0,0
Exp/Cntr=0.3,0.1

Type RM Length L Ch R = 1 ,3500    ,496.8,500,504.2
XS GIS Cut Line= 6
1662303.91476133439431.6857390111662403.60189793439418.794032499
 1662491.5016565439417.8668690031662566.49625717439418.750069335
1662741.48442426439420.8081360911662922.69928493439423.208065674
#Sta/Elev= 30
       0  1080.8     8.3 1079.79    24.4 1073.81    36.5 1064.42    48.6 1058.31
    76.8 1050.28     101  1030.7     117 1012.61     145 1001.28     161  990.25
     173  984.71     213  951.86     229  943.07     241  933.69  291.49928.8568
     301  928.18   322.1  928.79   356.4  942.77     397   962.4   433.1  994.67
   453.1 1015.11   465.1 1028.75   477.8 1047.42   485.1 1055.22   501.1 1062.09
   519.7 1073.23   545.1 1082.38   593.1  1112.7   613.1 1127.38   619.7  1129.9
#Mann= 3 ,-1,0
       0      .1       0  291.49    .045       0   322.1      .1       0
Bank Sta=291.49,322.1
XS Rating Curve= 0 ,0
Exp/Cntr(USF)=0,0
Exp/Cntr=0.3,0.1

Type RM Length L Ch R = 1 ,3000    ,510.5,498.9,483.6
XS GIS Cut Line= 6
1662336.11023501439867.5267308351662431.56706509 439872.43977876
1662519.80999884439880.2809704241662593.15827735439896.027001917
1662690.42711167439919.2385696771662939.67858167439978.717453346
#Sta/Elev= 30
       0  1086.9       4 1083.39      28 1077.28    44.1 1064.61    64.1 1056.97
    99.9 1029.72   140.3  993.52   164.4  973.75   188.6  955.62     209  943.92
   218.3  940.51   233.6  928.08   237.7  926.41   294.9   922.6   311.6  920.76
  326.34922.5751   352.7  940.56   360.9  948.09   373.3  952.62   381.5  957.88
   402.9  986.23   430.8 1013.52   455.5 1026.97   488.4 1051.37   500.7 1056.65
   513.1 1065.57   537.8 1074.81   554.2 1085.94   566.5  1087.8   615.4  1114.9
#Mann= 3 ,-1,0
       0      .1       0   294.9    .045       0  326.34      .1       0
Bank Sta=294.9,326.34
XS Rating Curve= 0 ,0
Exp/Cntr(USF)=0,0
Exp/Cntr=0.3,0.1

Type RM Length L Ch R = 1 ,2501    ,504.4,501.1,495.4
XS GIS Cut Line= 6
1662473.62111484440565.6608332541662669.48981759440400.473171502
1662746.02214484440335.6117526741662806.48691893440283.484232262
1662872.93363643440217.8341010961662943.41413851440146.255176008
#Sta/Elev= 30
       0 1088.33    14.2 1082.67    32.8  1070.4    45.1 1067.88    50.4 1064.52
      65 1049.18    81.8 1036.33   102.7  1017.2   121.8  992.08   164.4  962.69
   206.9  939.35   215.5  938.87   228.3  942.35   243.8  932.86   272.2  926.67
   283.6  922.17   291.1  916.95   301.6  915.33     318  916.94   340.3  917.15
     346  918.95   355.1  924.77   375.2  948.37   408.4  958.59     428  975.39
   449.9  989.08   489.3 1007.05   503.2 1015.49   591.3 1060.15   630.2 1072.73
#Mann= 3 ,-1,0
       0      .1       0   291.1    .045       0     318      .1       0
Bank Sta=291.1,318
XS Rating Curve= 0 ,0
Exp/Cntr(USF)=0,0
Exp/Cntr=0.3,0.1
